--- D112-00-00.prj (project) ---

Proj Title=D112-00-00
Current Plan=p02
Default Exp/Contr=.3,.1
English Units
Geom File=g05
Flow File=f01
Flow File=f06
Flow File=f04
Plan File=p06
Plan File=p02
Plan File=p04
Y Axis Title=Elevation
X Axis Title(PF)=Main Channel Distance
X Axis Title(XS)=Station
BEGIN DESCRIPTION:
Brays Bayou Watershed
Willow Waterhole Bayou
HCFCD Unit D112-00-00
Flood Hazard & Floodway Model
10, 2, 1, 0.2% Event
Filename D112.prj
Prepared by: Dodson & Associates, Inc.   Date: September 2003
Reviewed by:____________________	 Date:_________
STATUS (Final RAS, SVSQ)
FOR FLOOD HARZARD RECOVERY DATA ONLY,03/02/2004
Will Be Voided Upon Release of The Preliminary DFIRM
END DESCRIPTION:
DSS File=dss
DSS Export Rating Curves= 0
DSS Export Rating Curve Sorted= 0
DSS Export Volume Flow Curves= 0
DXF OffsetX= 0
DXF OffsetY= 0
DXF ScaleX= 1
DXF ScaleY= 10

--- D112-00-00.p02 (plan) ---

Plan Title=Floodway
Version=Version 3.0.1  Mar 2001
Short Identifier=Floodway0607
Geom File=g05
Flow File=f06
Subcritical Flow
K Sum by GR= 0
Std Step Tol= 0.01
Critical Tol= 0.01
Num of Std Step Trials= 20
Max Error Tol= 0.3
Flow Tol Ratio= 0.001
Split Flow NTrial= 30
Split Flow Tol= 0.02
Split Flow Ratio= 0.02
Log Output Level= 0
Friction Slope Method= 1
Unsteady Friction Slope Method= 2
Parabolic Critical Depth
Global Vel Dist= 0 , 0 , 0
Global Log Level= 0
CheckData=True
Encroach Param=-1 ,0,0, 2
Encroach River=D112-00-00
Encroach Reach=D112-00-00
Encroach Node=22325
       1    2046    2097
Encroach Node=21752
       1    2267    2328
Encroach Node=21164
       1    2275    2331
Encroach Node=20551
       1    2282    2340
Encroach Node=20273
       1    2264 2363.62
Encroach Node=20223
       1 2286.34 2361.57
Encroach Node=20201
       1 2273.04 2361.57
Encroach Node=20178
       1 2273.04 2346.86
Encroach Node=20123
       1 2274.86 2349.57
Encroach Node=20097
       1 2274.86 2363.62
Encroach Node=20071
       1 2282.55 2363.62
Encroach Node=20029
       1 2280.36    2369
Encroach Node=19789
       1 2198.64  2278.1
Encroach Node=18770
       1 2365.11 2445.34
Encroach Node=18277
       1 2348.18 2424.29
Encroach Node=18226
       1 2353.02 2425.98
Encroach Node=18197
       1 2353.02 2431.98
Encroach Node=18167
       1 2359.02 2431.98
Encroach Node=18125
       1 2349.84 2431.98
Encroach Node=17727
       1 2242.06 2305.74
Encroach Node=17323
       1 2140.93  2207.5
Encroach Node=16410
       1 1620.84 1708.37
Encroach Node=16158
       1 1998.96 2127.86
Encroach Node=16106
       1 2039.68 2130.68
Encroach Node=16082
       1 2039.68 2150.27
Encroach Node=16057
       1 2064.51 2150.27
Encroach Node=15937
       1 2112.85 2203.78
Encroach Node=15913
       1 2112.85 2235.58
Encroach Node=15888
       1 2147.85 2235.58
Encroach Node=15814
       1 2160.85 2248.58
Encroach Node=15667
       1 2283.82 2373.28
Encroach Node=14972
       1  1984.3 2070.79
Encroach Node=13959
       1 1622.02 1698.17
Encroach Node=12971
       1 1480.36 1592.97
Encroach Node=12115
       1 1475.39 1567.03
Encroach Node=10751
       1 1869.22  1968.7
Encroach Node=10059
       1 2250.68 2376.46
Encroach Node=9723
       1  2548.3 2676.98
Encroach Node=9642
       1 2561.23 2703.18
Encroach Node=9564
       1 2561.23 2703.18
Encroach Node=9486
       1 2563.13 2681.97
Encroach Node=9421
       1 2562.08 2667.69
Encroach Node=7801
       1 2408.11 2486.02
Encroach Node=7728
       1 2410.61 2491.76
Encroach Node=7704
       1 2410.61 2495.79
Encroach Node=7680
       1 2417.88 2495.79
Encroach Node=7649
       1 2411.96  2497.5
Encroach Node=7625
       1  2404.6  2497.5
Encroach Node=7601
       1  2404.6 2487.42
Encroach Node=7534
       1 2412.27 2490.18
Encroach Node=7144
       1 2389.05 2500.02
Encroach Node=5973
       1 1880.87 1988.04
Encroach Node=5893
       1 1882.49 1989.66
Encroach Node=5872
       1 1882.49 1991.23
Encroach Node=5850
       1 1884.06 1991.23
Encroach Node=5821
       1 1880.55 1987.72
Encroach Node=5354
       1 1929.08 2021.08
Encroach Node=4828
       1 2095.84 2193.31
Encroach Node=4468
       1 1987.77  2081.8
Encroach Node=3922
       1 1977.53 2077.28
Encroach Node=3845
       1 1989.74 2089.49
Encroach Node=3796
       1 1989.74 2097.49
Encroach Node=3746
       1 1990.65 2097.49
Encroach Node=3609
       1 1967.42 2067.17
Encroach Node=2955
       1 1566.39 1670.36
Encroach Node=1723
       1   906.9 1027.79
Encroach Node=1669
       1  922.84 1058.17
Encroach Node=1508
       1  922.84 1150.37
Encroach Node=1346
       1 1048.21 1150.37
Encroach Node=1304
       1 1048.21 1150.37
Encroach Node=679
       1  528.72   601.8
Encroach Reach=D112-00-00_0007
Encroach Node=22325
       1    2046    2097
Encroach Node=21752
       1    2267    2328
Encroach Node=21164
       1    2275    2331
Encroach Node=20551
       1    2282    2340
Encroach Node=20273
       1    2264 2363.62
Encroach Node=20223
       1 2286.34 2361.57
Encroach Node=20201
       1 2273.04 2361.57
Encroach Node=20178
       1 2273.04 2346.86
Encroach Node=20123
       1 2274.86 2349.57
Encroach Node=20097
       1 2274.86 2363.62
Encroach Node=20071
       1 2282.55 2363.62
Encroach Node=20029
       1 2280.36    2369
Encroach Node=19789
       1 2198.64  2278.1
Encroach Node=18770
       1 2365.11 2445.34
Encroach Node=18277
       1 2348.18 2424.29
Encroach Node=18226
       1 2353.02 2425.98
Encroach Node=18197
       1 2353.02 2431.98
Encroach Node=18167
       1 2359.02 2431.98
Encroach Node=18125
       1 2349.84 2431.98
Encroach Node=17727
       1 2242.06 2305.74
Encroach Node=17323
       1 2140.93  2207.5
Encroach Node=16410
       1 1620.84 1708.37
Encroach Node=16158
       1 1998.96 2127.86
Encroach Node=16106
       1 2039.68 2130.68
Encroach Node=16082
       1 2039.68 2150.27
Encroach Node=16057
       1 2064.51 2150.27
Encroach Node=15937
       1 2112.85 2203.78
Encroach Node=15913
       1 2112.85 2235.58
Encroach Node=15888
       1 2147.85 2235.58
Encroach Node=15814
       1 2160.85 2248.58
Encroach Node=15667
       1 2283.82 2373.28
Encroach Node=14972
       1  1984.3 2070.79
Encroach Node=13959
       1 1622.02 1698.17
Encroach Node=12971
       1 1480.36 1592.97
Encroach Node=12115
       1 1475.39 1567.03
Encroach Node=10751
       1 1869.22  1968.7
Encroach Node=10059
       1 2250.68 2376.46
Encroach Node=9723
       1  2548.3 2676.98
Encroach Node=9642
       1 2561.23 2703.18
Encroach Node=9564
       1 2561.23 2703.18
Encroach Node=9486
       1 2563.13 2681.97
Encroach Node=9421
       1 2562.08 2667.69
Encroach Node=7801
       1 2408.11 2486.02
Encroach Node=7728
       1 2410.61 2491.76
Encroach Node=7704
       1 2410.61 2495.79
Encroach Node=7680
       1 2417.88 2495.79
Encroach Node=7649
       1 2411.96  2497.5
Encroach Node=7625
       1  2404.6  2497.5
Encroach Node=7601
       1  2404.6 2487.42
Encroach Node=7534
       1 2412.27 2490.18
Encroach Node=7144
       1 2389.05 2500.02
Encroach Node=5973
       1 1880.87 1988.04
Encroach Node=5893
       1 1882.49 1989.66
Encroach Node=5872
       1 1882.49 1991.23
Encroach Node=5850
       1 1884.06 1991.23
Encroach Node=5821
       1 1880.55 1987.72
Encroach Node=5354
       1 1929.08 2021.08
Encroach Node=4828
       1 2095.84 2193.31
Encroach Node=4468
       1 1987.77  2081.8
Encroach Node=3922
       1 1977.53 2077.28
Encroach Node=3845
       1 1989.74 2089.49
Encroach Node=3796
       1 1989.74 2097.49
Encroach Node=3746
       1 1990.65 2097.49
Encroach Node=3609
       1 1967.42 2067.17
Encroach Node=2955
       1 1566.39 1670.36
Encroach Node=1723
       1   906.9 1027.79
Encroach Node=1669
       1  922.84 1058.17
Encroach Node=1508
       1  922.84 1150.37
Encroach Node=1346
       1 1048.21 1150.37
Encroach Node=1304
       1 1048.21 1150.37
Encroach Node=679
       1  528.72   601.8
Computation Interval=1HOUR
Output Interval=1HOUR
Run HTab= 0
Run UNet= 0
Run PostProcess= 0
UNET Theta= 1
UNET ZTol= 0.02
UNET ZSATol= 0.1
UNET MxIter= 20
UNET MaxInSteps= 20
UNET DtIC= 0
UNET DtMin= 0
UNET MaxCRTS= 20
UNET WFStab= 2
UNET SFStab= 1
UNET WFX= 1
UNET SFX= 1
UNET Convert EG Bridges=-1
UNET Use Existing IB Tables=-1
Instantaneous Interval=1HOUR
Write IC File= 0
Write Velocity= 0
Write Detailed= 0

--- D112-00-00.p01 (plan) ---

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Plan Title=Plan 01
Short Identifier=SV-SQ
Geom File=g05
Flow File=f01
Encroach Param=-1 ,0,0, 0

--- D112-00-00.p04 (plan) ---

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Plan Title=Storage Routing
Short Identifier=Store_Rout
Geom File=g05
Flow File=f04
Encroach Param=-1 ,0,0, 0

--- D112-00-00.p06 (plan) ---

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Plan Title=FEMA Effective June 2007
Short Identifier=FEMAeff0607
Geom File=g05
Flow File=f01
Encroach Param=-1 ,0,0, 0
DSS File=dss

--- D112-00-00.f06 (steady flow) ---

Flow Title=Floodway
Version=Version 3.0.1  Mar 2001
Number of Profiles= 2
Profile Names=1PCT_100yr,1PCTFloodway_100yrFW
River Rch & RM=D112-00-00,D112-00-00_0007 ,22325
    1033    1033
River Rch & RM=D112-00-00,D112-00-00_0007 ,21752
    1182    1182
River Rch & RM=D112-00-00,D112-00-00_0007 ,21164
    1360    1360
River Rch & RM=D112-00-00,D112-00-00_0007 ,20551
    1533    1533
River Rch & RM=D112-00-00,D112-00-00_0007 ,20029
    1565    1565
River Rch & RM=D112-00-00,D112-00-00_0007 ,18125
    1565    1565
River Rch & RM=D112-00-00,D112-00-00_0007 ,15814
    1730    1730
River Rch & RM=D112-00-00,D112-00-00_0007 ,14972
    1981    1981
River Rch & RM=D112-00-00,D112-00-00_0007 ,13959
    2261    2261
River Rch & RM=D112-00-00,D112-00-00_0007 ,12971
    2536    2536
River Rch & RM=D112-00-00,D112-00-00_0007 ,12115
    3041    3041
River Rch & RM=D112-00-00,D112-00-00_0007 ,10751
    3628    3628
River Rch & RM=D112-00-00,D112-00-00_0007 ,9421
    4001    4001
River Rch & RM=D112-00-00,D112-00-00_0007 ,7144
    4321    4321
River Rch & RM=D112-00-00,D112-00-00_0007 ,5354
    4595    4595
River Rch & RM=D112-00-00,D112-00-00_0007 ,3922
    5050    5050
River Rch & RM=D112-00-00,D112-00-00_0007 ,1723
    5438    5438
Boundary for River Rch & Prof#=D112-00-00,D112-00-00_0007 , 1
Up Type= 0
Dn Type= 1
Dn Known WS=46.44
Boundary for River Rch & Prof#=D112-00-00,D112-00-00_0007 , 2
Up Type= 0
Dn Type= 1
Dn Known WS=46.44
DSS Import GetInterval= 0
DSS Import GetPeak= 0
DSS Import FillOption= 0

--- D112-00-00.f01 (steady flow) ---

Flow Title=FEMA Effective June 2007
Version=Version 3.0.1  Mar 2001
Number of Profiles= 4
Profile Names=10PCT_10yr,2PCT_50yr,1PCT_100yr,0.2PCT_500yr
River Rch & RM=D112-00-00,D112-00-00_0007 ,22325
      35     843    1033    1344
River Rch & RM=D112-00-00,D112-00-00_0007 ,21752
      95     962    1182    1578
River Rch & RM=D112-00-00,D112-00-00_0007 ,21164
     271    1103    1360    1865
River Rch & RM=D112-00-00,D112-00-00_0007 ,20551
     663    1240    1533    2151
River Rch & RM=D112-00-00,D112-00-00_0007 ,20029
    1027    1400    1565    2151
River Rch & RM=D112-00-00,D112-00-00_0007 ,18125
    1099    1400    1565    2020
River Rch & RM=D112-00-00,D112-00-00_0007 ,15814
    1199    1536    1730    2147
River Rch & RM=D112-00-00,D112-00-00_0007 ,14972
    1330    1761    1981    2464
River Rch & RM=D112-00-00,D112-00-00_0007 ,13959
    1473    2014    2261    2819
River Rch & RM=D112-00-00,D112-00-00_0007 ,12971
    1609    2262    2536    3168
River Rch & RM=D112-00-00,D112-00-00_0007 ,12115
    1886    2700    3041    3793
River Rch & RM=D112-00-00,D112-00-00_0007 ,10751
    2201    3208    3628    4519
River Rch & RM=D112-00-00,D112-00-00_0007 ,9421
    2413    3531    4001    5013
River Rch & RM=D112-00-00,D112-00-00_0007 ,7144
    2593    3807    4321    5439
River Rch & RM=D112-00-00,D112-00-00_0007 ,5354
    2747    4044    4595    5806
River Rch & RM=D112-00-00,D112-00-00_0007 ,3922
    3002    4435    5050    6417
River Rch & RM=D112-00-00,D112-00-00_0007 ,1723
    3218    4769    5438    6941
Boundary for River Rch & Prof#=D112-00-00,D112-00-00_0007 , 1
Up Type= 0
Dn Type= 3
Dn Slope=.0006
Boundary for River Rch & Prof#=D112-00-00,D112-00-00_0007 , 2
Up Type= 0
Dn Type= 3
Dn Slope=.0006
Boundary for River Rch & Prof#=D112-00-00,D112-00-00_0007 , 3
Up Type= 0
Dn Type= 3
Dn Slope=.0006
Boundary for River Rch & Prof#=D112-00-00,D112-00-00_0007 , 4
Up Type= 0
Dn Type= 3
Dn Slope=.0006
DSS Import GetInterval= 0
DSS Import GetPeak= 0
DSS Import FillOption= 0

--- D112-00-00.f04 (steady flow) ---

Flow Title=Storage Routing
Version=Version 3.0.1  Mar 2001
Number of Profiles= 8
Profile Names=.1,.2,.4,.6,.8,1.0,1.2,1.5
River Rch & RM=D112-00-00,D112-00-00_0007 ,22325
     155     310     620     930    1240    1550    1860    2325
River Rch & RM=D112-00-00,D112-00-00_0007 ,20029
     156     312     624     936    1248    1560    1872    2340
River Rch & RM=D112-00-00,D112-00-00_0007 ,18125
     153     306     612     918    1224    1530    1836    2295
River Rch & RM=D112-00-00,D112-00-00_0007 ,15814
     252     504    1008    1512    2016    2520    3024    3780
River Rch & RM=D112-00-00,D112-00-00_0007 ,12115
     362     724    1448    2172    2896    3620    4344    5430
River Rch & RM=D112-00-00,D112-00-00_0007 ,9421
     543    1086    2172    3258    4344    5430    6516    8145
Boundary for River Rch & Prof#=D112-00-00,D112-00-00_0007 , 1
Up Type= 0
Dn Type= 3
Dn Slope=.0006
Boundary for River Rch & Prof#=D112-00-00,D112-00-00_0007 , 2
Up Type= 0
Dn Type= 3
Dn Slope=.0006
Boundary for River Rch & Prof#=D112-00-00,D112-00-00_0007 , 3
Up Type= 0
Dn Type= 3
Dn Slope=.0006
Boundary for River Rch & Prof#=D112-00-00,D112-00-00_0007 , 4
Up Type= 0
Dn Type= 3
Dn Slope=.0006
Boundary for River Rch & Prof#=D112-00-00,D112-00-00_0007 , 5
Up Type= 0
Dn Type= 3
Dn Slope=.0006
Boundary for River Rch & Prof#=D112-00-00,D112-00-00_0007 , 6
Up Type= 0
Dn Type= 3
Dn Slope=.0006
Boundary for River Rch & Prof#=D112-00-00,D112-00-00_0007 , 7
Up Type= 0
Dn Type= 3
Dn Slope=.0006
Boundary for River Rch & Prof#=D112-00-00,D112-00-00_0007 , 8
Up Type= 0
Dn Type= 3
Dn Slope=.0006
DSS Import GetInterval= 0
DSS Import GetPeak= 0
DSS Import FillOption= 0

--- D112-00-00.g05 (geometry) ---

Geom Title=D112-00-00 June 2007
Version=Version 3.0.1  Mar 2001

River Reach=D112-00-00      ,D112-00-00_0007
Reach XY= 30
     3080395.471    13802165.174     3080794.689    13802042.537
     3082414.068    13800729.186      3083135.29    13800420.365
      3083455.03    13800436.853     3085129.683    13801035.823
     3085449.298    13801552.103     3085561.109    13801621.946
     3085904.452    13801678.097     3086393.755    13801639.253
     3086772.171     13801761.29     3087116.834    13801791.879
     3089325.117    13803482.054     3089735.048    13803490.379
      3089801.24     13803698.84        3090078.    13803802.821
     3090317.976    13804122.768     3090886.264    13804293.045
     3091664.084    13805033.589     3091703.378    13805266.295
     3091833.518    13805478.054       3092332.5    13805922.847
     3092913.143    13806674.316     3093164.196    13807276.779
     3094396.508    13808993.546     3094447.201      13809502.5
     3094280.081    13810256.284      3094294.98     13810961.91
     3094597.451    13811810.526     3094763.144      13812547.5

Type RM Length L Ch R = 1 ,22325   ,574.94,572.42,572.74
BEGIN DESCRIPTION:
22324.82-- Used Channel Survey from DAI 1997 report
END DESCRIPTION:
XS GIS Cut Line= 6
     3080833.104    13804152.689     3080825.641    13802375.782
     3080711.578    13802177.522     3080656.021    13802092.088
     3080501.051    13801513.052 3080558.667932813800518.6684026
#Sta/Elev= 30
       0   61.24  305.19   61.59  391.23   57.32  425.19   60.29  466.55   60.59
  903.39   59.17  993.77   56.65  1190.2   58.89  1370.2   56.19  1535.2    58.3
  1745.2   58.25 1844.16   56.23 1999.91   58.18  2035.5   55.29    2046    56.3
    2053    49.4    2063      49    2075    49.6    2097    58.1 2402.17   58.56
 2448.75   55.43 2510.86   56.45 2603.79   50.96 2666.14   56.93 2723.07   58.18
 3163.29   59.63 3291.16   58.02 3433.19   59.76 3589.41   57.48 3703.03   59.55
#Mann= 3 , 0 , 0
       0     .15       0    2046     .04       0    2097     .15       0
#XS Ineff= 2 , 0
       0    1990            2145       0
Permanent Ineff=
       T       T
#Block Obstruct= 1 ,-1
 2403.15 2699.76   57.69
Bank Sta=2046,2097
XS Rating Curve= 0
Exp/Cntr=.3,.1

Type RM Length L Ch R = 1 ,21752   ,582.94,588.53,593.95
BEGIN DESCRIPTION:
21752.40--Used Channel Survey from DAI 1997 report
END DESCRIPTION:
XS GIS Cut Line= 6
     3081269.965    13804034.136     3081261.427    13802001.176
     3081147.364    13801802.916     3081091.807    13801717.483
     3080936.837    13801138.446     3081059.688    13799018.202
#Sta/Elev= 30
       0   60.76  186.64    60.9  246.64   58.45  291.64   61.05  396.64    61.7
  531.64   58.34  636.64   60.95 1206.65   57.09 1836.65   56.01 1971.65   58.33
 2090.98   55.95  2204.5   58.25    2267    56.6    2287    47.6    2293    47.4
    2328    57.3 3049.77   58.71 3149.19   56.39 3359.64   59.26 3461.64   56.43
 3546.85   59.49 3703.07   59.41  3750.3   57.11 3825.42   60.09 4058.13   57.66
 4114.94   60.05  4351.3   58.43 4907.23   60.75 4952.31   58.56 5086.83   61.02
#Mann= 3 , 0 , 0
       0     .15       0    2267     .04       0    2328     .15       0
#XS Ineff= 2 , 0
       0    2230            2363       0
Permanent Ineff=
       T       T
Bank Sta=2267,2328
XS Rating Curve= 0
Exp/Cntr=.3,.1

Type RM Length L Ch R = 1 ,21164   ,567.48,612.94,603.54
BEGIN DESCRIPTION:
21163.86--Used Channel Survey from DAI 1997 report
END DESCRIPTION:
XS GIS Cut Line= 6
     3081723.181    13803659.531     3081714.643    13801626.571
      3081600.58    13801428.311     3081545.023    13801342.877
     3081390.053    13800763.841     3081512.905    13798643.596
#Sta/Elev= 30
       0   61.83   97.03   61.57  157.03   58.61  247.03   61.73  387.98   61.43
  457.04   58.52  667.04   61.12  832.04   57.33  982.04   60.04 1141.15   56.48
 1222.04   58.76 1342.04   58.87 1417.04    56.3 1547.86    58.6 1894.32   58.56
 2097.43   55.33 2204.96   58.65    2275    55.2    2292    47.3    2300    46.5
    2331    56.2 2876.21    58.1 3074.56   55.72 3119.64   58.06 3375.06   57.33
 3465.21   59.32 3970.24   57.96 4036.17   60.11 4268.49   58.45 5086.83   61.45
#Mann= 3 , 0 , 0
       0     .15       0    2275     .04       0    2331     .15       0
#XS Ineff= 2 , 0
       0    2235            2365       0
Permanent Ineff=
       T       T
Bank Sta=2275,2331
XS Rating Curve= 0
Exp/Cntr=.3,.1

Type RM Length L Ch R = 1 ,20551   ,242.6,278.3,272.63
BEGIN DESCRIPTION:
20550.92--Used Channel Survey from DAI 1997 report
END DESCRIPTION:
XS GIS Cut Line= 6
     3082198.187    13803276.214     3082189.649    13801243.254
     3082075.586    13801044.994      3082020.03     13800959.56
     3081865.059    13800380.524     3081987.911    13798260.279
#Sta/Elev= 30
       0   60.63   43.71   58.31  369.58   62.33  655.79   61.23  718.72   58.43
  778.72      61 1183.01   60.78 1303.51   58.39 1378.73   58.19 1393.73   59.36
 1618.73   56.22 1903.73   57.33 1993.73    59.3 2247.28   57.56    2282    55.7
    2300    47.1    2308    45.9    2316    46.9    2340    55.7 2370.93   57.71
 2617.38   55.23 2871.81   55.65 3100.76   58.15 3862.56   58.11 3907.64   59.63
 4568.75   60.48  4634.6   61.67 4824.17   59.57 4914.32   61.45 5086.83   61.43
#Mann= 3 , 0 , 0
       0     .15       0    2282     .04       0    2340     .15       0
#XS Ineff= 2 , 0
       0    2240            2372       0
Permanent Ineff=
       T       T
Bank Sta=2282,2340
XS Rating Curve= 0
Exp/Cntr=.3,.1

Type RM Length L Ch R = 1 ,20273   ,45.17,50.09,49.96
BEGIN DESCRIPTION:
20272.61--u/s approach Hillcroft West bridge;  channel copied from 20071
END DESCRIPTION:
XS GIS Cut Line= 6
     3082422.673    13803111.963     3082414.135    13801079.003
     3082300.072    13800880.743     3082244.515     13800795.31
     3082089.545    13800216.273     3082212.396    13798096.029
#Sta/Elev= 30
       0   58.76  314.47   59.47  566.67   58.06  777.56   59.99   928.2   60.53
 1033.64   59.62 1093.89   60.72  1214.4   60.43 1259.47    59.4 1304.47   60.33
 1394.48   60.05 1454.48    56.8 1499.48   60.02 1514.48   60.25 1574.48   59.47
 1739.48   60.75 2056.31    55.7 2182.03   58.01    2264   57.63 2278.55   56.58
 2300.79   45.48 2304.79   45.18 2363.62   57.42 2495.93   57.34 2542.51   55.61
 2697.79   57.57 2988.34   57.73 3215.58   56.51 3471.22   58.06 5086.83   61.36
#Mann= 3 , 0 , 0
       0     .15       0    2264     .04       0 2363.62     .15       0
#XS Ineff= 2 , 0
       0    2260            2370       0
Permanent Ineff=
       T       T
Bank Sta=2264,2363.62
XS Rating Curve= 0
Exp/Cntr=.5,.3

Type RM Length L Ch R = 1 ,20223   ,39.75,44.08,43.97
BEGIN DESCRIPTION:
20222.52--u/s face Hillcroft West bridge;  channel copied from 20071
END DESCRIPTION:
XS GIS Cut Line= 6
     3082464.485    13803084.373     3082455.947    13801051.413
     3082341.884    13800853.153     3082286.327     13800767.72
     3082131.357    13800188.683     3082251.422    13798114.897
#Sta/Elev= 30
       0   59.23  271.03   59.69  616.88   58.38  691.88   59.26  856.88    59.3
 1400.78   56.68 1486.89   57.72 1521.29   56.89 1536.35   57.53 1741.89   57.81
 1958.13   57.14 2032.98   56.16 2140.15   56.71 2286.34   55.54 2306.79   45.48
 2310.79   45.18 2361.57   56.06 2365.62   56.91    2545   55.73 3129.49   57.31
  3309.8   57.02 3419.73   57.89 3448.13   57.23 3685.42   59.08 3959.43   58.81
    4031   57.88 4712.18   61.23 4982.04   61.53 5007.63   60.88 5040.29   61.54
#Mann= 3 , 0 , 0
       0     .15       0 2286.34     .04       0 2361.57     .15       0
#XS Ineff= 2 , 0
       0    2264            2359       0
Permanent Ineff=
       T       T
Bank Sta=2286.34,2361.57
XS Rating Curve= 0
Exp/Cntr=.5,.3

Type RM Length L Ch R = 3 ,20201   ,,,
BEGIN DESCRIPTION:
Hillcroft West (U) Bridge
END DESCRIPTION:
Bridge Culvert--1,0,-1,-1, 0
Deck Dist Width WeirC Skew NumUp NumDn MinLoCord MaxHiCord MaxSubmerge Is_Ogee
5,34,2.6,0, 7, 7, , , .95, 0, 0,0,,
 2192.51 2289.94 2289.94 2320.29 2350.63 2350.63 2494.89
   56.17   56.53   56.53   56.47   56.53   56.53   55.98
     -.2     -.2   54.85   54.79   54.85     -.2     -.2
 2183.01 2280.44 2280.44 2310.79 2341.13 2341.13 2485.39
   56.17   56.53   56.53   56.47   56.53   56.53   55.98
     -.2     -.2   54.85   54.79   54.85     -.2     -.2
Pier Skew, UpSta & Num, DnSta & Num=  ,2300.17, 2 ,2290.67, 2 , 0 , 0 , 0 ,,
    1.67    1.67
       0   54.85
    1.67    1.67
       0   54.85
Pier Skew, UpSta & Num, DnSta & Num=  ,2325.4, 2 ,2315.9, 2 , 0 , 0 , 0 ,,
    1.67    1.67
       0   54.85
    1.67    1.67
       0   54.85
BR Coef=-1 , 1 , 1 ,1.05, 0 ,,,.8,-1,1.2,0,
WSPro=,,,, 1 ,,,, 0 ,,,, 0 ,,,,-1 ,-1 ,-1 , 0 , 0 , 0 , 0 , 0
BC Design=,, 0 ,, 0 ,,,,,,

Type RM Length L Ch R = 1 ,20178   ,49.69,55.1,54.96
BEGIN DESCRIPTION:
20178.44--d/s face Hillcroft West bridge;  channel copied from 20071
END DESCRIPTION:
XS GIS Cut Line= 6
      3082501.28    13803060.103     3082492.742    13801027.143
     3082378.679    13800828.883     3082323.122     13800743.45
     3082168.152    13800164.413     3082285.763      13798131.5
#Sta/Elev= 30
       0   58.79  322.61    59.6  526.04   58.21  622.61   58.23  787.61   59.28
  857.43   58.56 1188.83    57.9 1264.14   57.01 1279.21   57.55 1761.24   57.73
 2171.01   56.17 2273.04   55.18 2279.46   54.31 2297.29   45.48 2301.29   45.18
 2346.86   54.98 2395.66   56.13 2519.56   56.31 2566.46   55.59 2814.91   57.18
 3060.11   57.01 3075.13   56.31 3191.48   57.34 3631.06   58.54  3674.4    59.2
 4043.68   58.68 4367.29   59.39 4441.38   60.15 4652.77   59.72 4999.34   60.58
#Mann= 3 , 0 , 0
       0     .15       0 2273.04     .04       0 2346.86     .15       0
#XS Ineff= 2 , 0
       0    2263            2355       0
Permanent Ineff=
       T       T
Bank Sta=2273.04,2346.86
XS Rating Curve= 0
Exp/Cntr=.5,.3

Type RM Length L Ch R = 1 ,20123   ,49.47,52.31,53.06
BEGIN DESCRIPTION:
20123.34--u/s face Hillcroft East bridge;  channel copied from 20071
END DESCRIPTION:
XS GIS Cut Line= 6
     3082547.273    13803029.753     3082538.735    13800996.793
     3082424.672    13800798.533     3082369.115      13800713.1
     3082214.145    13800134.063     3082328.692    13798152.255
#Sta/Elev= 30
       0   61.05  262.26   60.28  472.26   58.12  539.75   58.98  772.26    59.2
 1503.81   57.21 1729.76   57.94 1970.77   56.37 2035.45   58.51 2101.38   56.56
 2257.13   56.22 2274.86   55.39 2294.79   45.48 2298.79   45.18 2349.57   56.06
 2581.27   55.84 2991.36   57.25 3089.81   56.28 3374.87   58.14 3450.41    57.7
 3480.46    58.8 3559.53   58.99 3600.66   57.99 3658.95   59.16 3780.96   59.67
 3961.26   58.92 4141.56   60.03 4562.26   59.55 4837.89   61.32 4948.15   61.06
#Mann= 3 , 0 , 0
       0     .15       0 2274.86     .04       0 2349.57     .15       0
#XS Ineff= 2 , 0
       0    2262            2360       0
Permanent Ineff=
       T       T
Bank Sta=2274.86,2349.57
XS Rating Curve= 0
Exp/Cntr=.5,.3

Type RM Length L Ch R = 3 ,20097   ,,,
BEGIN DESCRIPTION:
Hillcroft East (D) Bridge
END DESCRIPTION:
Bridge Culvert--1,0,-1,-1, 0
Deck Dist Width WeirC Skew NumUp NumDn MinLoCord MaxHiCord MaxSubmerge Is_Ogee
9,34,2.6,0, 7, 7, , , .95, 0, 0,0,,
 2267.13 2278.36 2278.36 2308.29 2338.21 2338.21 2400.45
   56.22   56.43   56.43   56.33   56.42   56.42   56.26
     -.2     -.2   54.73   54.63   54.72     -.2     -.2
 2277.13 2287.36 2287.36 2317.79 2348.21 2348.21 2410.45
   56.22   56.43   56.43   56.33   56.42   56.42   56.26
     -.2     -.2   54.73   54.63   54.72     -.2     -.2
Pier Skew, UpSta & Num, DnSta & Num=  ,2290.31, 2 ,2300.31, 2 , 0 , 0 , 0 ,,
    1.67    1.67
       0   54.85
    1.67    1.67
       0   54.85
Pier Skew, UpSta & Num, DnSta & Num=  ,2309.26, 2 ,2319.26, 2 , 0 , 0 , 0 ,,
    1.67    1.67
       0   54.85
    1.67    1.67
       0   54.85
BR Coef=-1 , 1 , 1 ,1.05, 0 ,,,.8,-1,1.2,0,
WSPro=,,,, 1 ,,,, 0 ,,,, 0 ,,,,-1 ,-1 ,-1 , 0 , 0 , 0 , 0 , 0
BC Design=,, 0 ,, 0 ,,,,,,

Type RM Length L Ch R = 1 ,20071   ,42.52,42.49,42.27
BEGIN DESCRIPTION:
20071.03--d/s face Hillcroft East bridge; surveyed channel
END DESCRIPTION:
XS GIS Cut Line= 6
     3082593.083    13803005.126     3082584.545    13800972.166
     3082470.482    13800773.906     3082414.925    13800688.472
     3082259.955    13800109.436     3082376.688    13798163.885
#Sta/Elev= 30
       0   62.52  342.63   62.37   393.7   61.45  432.63   58.37  447.63   58.24
  484.08    61.3  597.63    60.9  642.63   61.73 1242.64   58.31 1317.64   56.51
 2067.16   60.15 2217.56   59.07 2282.55   56.58 2304.79   45.48 2308.79   45.18
 2363.62   56.91 2431.91   57.37 2524.12   55.65 2571.66   57.09 2726.94   57.78
 3050.12   57.08 3477.62   59.83 3561.04   58.03  3605.2   59.89 3690.26   60.61
 4162.12   61.68 4413.26   60.74 4477.69   59.62 4753.49   61.82 4912.08   61.33
#Mann= 3 , 0 , 0
       0     .15       0 2282.55     .04       0 2363.62     .15       0
#XS Ineff= 2 , 0
       0    2265            2380       0
Permanent Ineff=
       T       T
Bank Sta=2282.55,2363.62
XS Rating Curve= 0
Exp/Cntr=.5,.3

Type RM Length L Ch R = 1 ,20029   ,245.5,239.97,285.03
BEGIN DESCRIPTION:
20028.55--d/s exit Hillcroft East bridge;  channel copied from 20071
END DESCRIPTION:
XS GIS Cut Line= 6
      3082632.48    13802989.353     3082623.942    13800956.393
     3082509.879    13800758.133     3082454.322      13800672.7
     3082299.352    13800093.663      3082409.14    13798191.149
#Sta/Elev= 30
       0   63.17  341.86   62.72  371.86   62.24  431.86   58.18  461.86   61.63
  669.69   62.49 1211.86   61.27 1271.86   60.37 1316.86    57.1 1391.87    60.3
 1526.87    60.7 2227.83   59.64 2280.36   57.16 2304.79   45.48 2308.79   45.18
    2369   57.92 2462.17   57.83 2508.75   55.51 2570.86   57.23 2664.03   57.72
 3213.34   58.38 3454.83   60.11 3515.11   59.86 3545.16   58.14 3605.26   60.71
  4193.5   61.54 4506.02   59.66 4596.91   61.42 4732.13   62.08 4868.71   61.37
#Mann= 3 , 0 , 0
       0     .15       0 2280.36     .04       0    2369     .15       0
#XS Ineff= 2 , 0
       0    2267            2375       0
Permanent Ineff=
       T       T
Bank Sta=2280.36,2369
XS Rating Curve= 0
Exp/Cntr=.3,.1

Type RM Length L Ch R = 1 ,19789   ,783.04,1018.76,1060.95
BEGIN DESCRIPTION:
 19788.57--surveyed channel
END DESCRIPTION:
XS GIS Cut Line= 5
     3082880.026     13802793.84     3082939.819    13801290.475
     3082711.276    13800656.277     3082676.812    13800563.015
     3082805.992    13798383.018
#Sta/Elev= 30
       0   60.27  161.47   60.36  221.52   57.84  330.92    60.7  518.61   58.57
  641.85   60.75  806.98   58.06  897.05   60.24 1122.23    58.2 1211.62   60.23
 1547.19   59.65 1746.61   56.81  2007.3   55.65 2102.97   57.63 2198.64   55.58
 2229.75   45.04  2278.1   57.04 2458.79   55.79 2898.68   58.47 3029.93   57.06
 3210.25   60.06 3330.46   58.55 3375.54   60.69 3570.88   60.63 3615.96   58.53
  3811.3   61.02 3931.51   59.03 4126.85    61.6 4232.04   59.17 4461.92   62.14
#Mann= 3 , 0 , 0
       0     .15       0 2198.64     .04       0  2278.1     .15       0
#XS Ineff= 2 , 0
       0    2168            2280       0
Permanent Ineff=
       T       T
Bank Sta=2198.64,2278.1
XS Rating Curve= 0
Exp/Cntr=.3,.1

Type RM Length L Ch R = 1 ,18770   ,483.25,492.45,491.67
BEGIN DESCRIPTION:
 18769.81--surveyed channel
END DESCRIPTION:
XS GIS Cut Line= 5
     3083538.465    13802894.727     3083645.221    13800548.978
     3083677.572     13800457.36     3083933.578    13799403.488
     3083955.552    13799021.687
#Sta/Elev= 30
       0   58.57   52.28   61.08  202.44   61.06  277.51   59.29  352.59   61.12
  577.82   59.72   757.6   61.23  893.15   58.86  953.21   60.57 1193.46   59.07
 1288.99   60.21 1493.77   58.04 1598.88   59.16 1820.38    57.1 1869.16   55.26
 1974.27   57.21 2124.42   56.63 2179.43   55.07 2244.55   57.06 2365.11   54.35
 2392.98   44.32 2402.47   45.09 2445.34   55.46 2494.84   56.77 2606.61   54.24
 2753.92   57.84 3488.39   60.27 3661.06   59.33 3721.16   61.03 3912.29   60.98
#Mann= 3 , 0 , 0
       0     .15       0 2365.11     .04       0 2445.34     .15       0
#XS Ineff= 2 , 0
       0    2334            2450       0
Permanent Ineff=
       T       T
Bank Sta=2365.11,2445.34
XS Rating Curve= 0
Exp/Cntr=.3,.1

Type RM Length L Ch R = 1 ,18277   ,49.1,51.41,51.27
BEGIN DESCRIPTION:
18277.36--u/s approach Landsdowne bridge; channel copied from 18167
END DESCRIPTION:
XS GIS Cut Line= 5
     3084012.735    13803050.712     3084119.491    13800704.963
     3084139.914    13800610.417     3084407.848    13799559.473
     3084429.822    13799177.672
#Sta/Elev= 30
       0   61.53   58.27   61.05  118.33   58.04  165.62   60.48  352.32   60.68
  424.13   58.16  508.74   61.01  613.85   61.12  703.94   58.24     764   60.33
   959.2   60.47 1019.27   57.64 1084.78   59.84 1304.56    57.9 1364.62    59.6
 1484.75   59.76 1604.87   56.72 1731.07   57.63 1917.77   54.53 2047.03   55.99
 2190.48   54.42 2250.54   56.46 2348.18   56.14  2386.2   43.04 2424.29   56.18
 2525.31   57.19 2572.78   54.63  3299.3   58.92 3485.06   56.94  3911.9   58.75
#Mann= 3 , 0 , 0
       0     .15       0 2348.18     .04       0 2424.29     .15       0
#XS Ineff= 2 , 0
       0    2331            2430       0
Permanent Ineff=
       T       T
Bank Sta=2348.18,2424.29
XS Rating Curve= 0
Exp/Cntr=.5,.3

Type RM Length L Ch R = 1 ,18226   ,56.36,58.81,58.61
BEGIN DESCRIPTION:
18225.95--u/s face Landsdowne bridge; channel copied from 18167
END DESCRIPTION:
XS GIS Cut Line= 5
     3084060.735    13803069.712     3084167.491    13800723.963
     3084187.914    13800629.417     3084455.848    13799578.473
     3084477.822    13799196.672
#Sta/Elev= 30
       0   61.49   92.31   60.34  122.34   57.69  238.39   60.31   377.6   59.84
  425.09   57.75   496.9   60.13  640.52   60.28  722.96   57.71  899.03   60.29
 1038.29   57.82 1113.36    59.8 1293.55   59.07 1329.89   57.45 1518.78   59.28
 1623.89   56.64 1759.03   57.34  1924.2   54.87 2353.02   55.35  2388.2   43.04
 2425.98   55.93 2622.32   54.66 2844.97    56.9 2916.44   55.72 3461.72   58.02
 3511.06   56.97  3565.1   59.06 3721.38   59.61 3790.87   58.33  3911.9   60.36
#Mann= 3 , 0 , 0
       0     .15       0 2353.02     .04       0 2425.98     .15       0
#XS Ineff= 2 , 0
       0    2333            2430       0
Permanent Ineff=
       T       T
Bank Sta=2353.02,2425.98
XS Rating Curve= 0
Exp/Cntr=.5,.3

Type RM Length L Ch R = 3 ,18197   ,,,
BEGIN DESCRIPTION:
Landsdowne Bridge
END DESCRIPTION:
Bridge Culvert--1,0,-1,-1, 0
Deck Dist Width WeirC Skew NumUp NumDn MinLoCord MaxHiCord MaxSubmerge Is_Ogee
9,40,2.6,0, 7, 7, , , .95, 0, 0,0,,
    2330 2359.65 2359.65  2389.2 2417.74 2417.74    2434
   56.04   56.04   56.04   56.09   56.05   56.05   56.05
     -.2     -.2   54.45    54.5   54.46     -.2     -.2
    2336 2365.65 2365.65  2395.2 2423.74 2423.74    2440
   56.04   56.04   56.04   56.09   56.05   56.05   56.05
     -.2     -.2   54.45    54.5   54.46     -.2     -.2
Pier Skew, UpSta & Num, DnSta & Num=  ,2378.68, 2 ,2384.68, 2 , 0 , 0 , 0 ,,
    1.69    1.69
       0    54.6
    1.69    1.69
       0    54.6
Pier Skew, UpSta & Num, DnSta & Num=  ,2397.71, 2 ,2403.71, 2 , 0 , 0 , 0 ,,
    1.69    1.69
       0    54.6
    1.69    1.69
       0    54.6
BR Coef=-1 , 1 , 1 ,1.05, 0 ,,,.8,-1,1.2,0,
WSPro=,,,, 1 ,,,, 0 ,,,, 0 ,,,,-1 ,-1 ,-1 , 0 , 0 , 0 , 0 , 0
BC Design=,, 0 ,, 0 ,,,,,,

Type RM Length L Ch R = 1 ,18167   ,40.72,42.49,42.34
BEGIN DESCRIPTION:
18167.13--d/s face Landsdowne bridge; surveyed channel
END DESCRIPTION:
XS GIS Cut Line= 5
     3084115.891    13803090.314     3084222.648    13800744.564
      3084243.07    13800650.019     3084511.005    13799599.074
     3084532.978    13799217.273
#Sta/Elev= 30
       0   61.44  104.77   60.42  142.96   57.71  219.66   59.33 1013.86   59.38
 1043.89   58.36 1196.27   59.44 1368.62   58.04 1419.28   59.29 2170.06   54.39
  2305.2   56.06 2359.02   55.35  2394.2   43.04 2431.98   55.93 2488.78   56.61
 2597.14   54.72 2659.06   56.79  2865.9   57.69 2939.91   56.16 2984.14    57.8
  3092.5    58.2 3211.28   56.58 3262.77   58.72 3470.31   58.69 3519.66   57.25
 3603.41    59.6 3674.45   58.83 3751.41   59.89 3816.52   58.43  3911.9   60.25
#Mann= 3 , 0 , 0
       0     .15       0 2359.02     .04       0 2431.98     .15       0
#XS Ineff= 2 , 0
       0    2336            2435       0
Permanent Ineff=
       T       T
Bank Sta=2359.02,2431.98
XS Rating Curve= 0
Exp/Cntr=.5,.3

Type RM Length L Ch R = 1 ,18125   ,366.61,397.34,388.66
BEGIN DESCRIPTION:
18124.65--d/s exit Landsdowne bridge; channel copied from 18167
END DESCRIPTION:
XS GIS Cut Line= 5
     3084155.735    13803105.212     3084262.491    13800759.463
     3084282.914    13800664.917     3084550.848    13799613.973
     3084572.822    13799232.172
#Sta/Elev= 30
       0   61.62   97.81   60.51  157.88   57.91  232.95   60.71  848.59   61.48
 1229.84   60.71 1358.56   58.05 1404.16   59.87 1509.27   59.84 2120.27    56.1
 2192.08   54.32 2349.84   56.32 2359.02   55.35  2394.2   43.04 2431.98   55.93
 2549.34   56.22 2611.02   54.66 2672.69    56.8 2798.27   57.77 2944.06   56.28
 3030.17   57.99 3178.43    58.1 3215.43   56.49 3264.77   58.38 3401.99   58.72
 3525.82   57.12  3608.2   59.31 3721.25   60.17 3841.45   58.63  3911.9   60.22
#Mann= 3 , 0 , 0
       0     .15       0 2349.84     .04       0 2431.98     .15       0
#XS Ineff= 2 , 0
       0    2341            2435       0
Permanent Ineff=
       T       T
Bank Sta=2349.84,2431.98
XS Rating Curve= 0
Exp/Cntr=.3,.1

Type RM Length L Ch R = 1 ,17727   ,321.33,404.5,448.75
BEGIN DESCRIPTION:
 17727.31--surveyed channel
END DESCRIPTION:
XS GIS Cut Line= 5
     3084424.029     13803097.66     3084636.399    13800890.017
     3084658.485    13800792.883     3084809.576    13800090.904
     3084850.117    13799371.304
#Sta/Elev= 30
       0   59.86  165.92   57.92  316.61   60.85  452.24   58.19  587.86   61.17
  693.35   60.87  738.55    58.1   813.9   61.16  976.14   61.02 1039.94   58.45
 1158.06   60.99 1350.52   58.24 1386.53   60.16 1642.71   59.16 1748.19   55.06
 1898.89   57.15 2004.37   56.02 2051.61   53.04 2109.85   55.04 2242.06   54.57
 2266.92   43.44 2273.43   42.96 2279.98   43.71 2305.74   55.16 2783.26   57.28
 2906.01   55.68 3065.21   57.99 3209.18   56.63 3314.35   58.87 3756.24   59.84
#Mann= 3 , 0 , 0
       0     .15       0 2242.06     .04       0 2305.74     .15       0
#XS Ineff= 2 , 0
       0    2219            2310       0
Permanent Ineff=
       T       T
Bank Sta=2242.06,2305.74
XS Rating Curve= 0
Exp/Cntr=.3,.1

Type RM Length L Ch R = 1 ,17323   ,798.97,912.78,584.32
BEGIN DESCRIPTION:
 17322.81--surveyed channel
END DESCRIPTION:
XS GIS Cut Line= 6
     3084781.776     13803110.31     3084844.651    13801469.853
     3085012.365    13801020.905     3085045.382    13800927.223
     3085229.034    13800410.664     3085254.527    13799566.827
#Sta/Elev= 30
       0   60.93   87.87    60.7  132.91   58.33  234.72   61.06  448.14   59.22
  639.51   61.14  733.35   58.77  823.41   61.04  1044.3    59.5 1198.69   61.17
 1333.44   58.43 1434.64   60.04 1579.21   58.82 1665.52   55.37 1789.48   57.26
 1969.76   54.34 2078.44   56.18 2140.93   54.38 2160.68    47.5 2165.06   43.84
 2172.69   42.95  2207.5   54.59 2256.42   56.16 2374.36   53.93 2671.01   56.28
 2931.72   54.71 2993.42   56.69 3241.05   55.83 3532.39      57  3612.7   59.05
#Mann= 3 , 0 , 0
       0     .15       0 2140.93     .04       0  2207.5     .15       0
#XS Ineff= 2 , 0
       0    2109            2215       0
Permanent Ineff=
       T       T
Bank Sta=2140.93,2207.5
XS Rating Curve= 0
Exp/Cntr=.3,.1

Type RM Length L Ch R = 1 ,16410   ,331.87,252.36,241.34
BEGIN DESCRIPTION:
 16410.04--surveyed channel
END DESCRIPTION:
XS GIS Cut Line= 6
     3085426.404    13803281.845     3085451.122    13802033.615
     3085580.388    13801697.804     3085619.865    13801605.733
      3085442.58    13800880.466      3085503.05    13799686.982
#Sta/Elev= 30
       0   59.87  184.38   60.45   289.4   58.31  348.61   60.25  525.15   60.49
  574.46    58.6  634.47   60.33  760.53   60.63  889.52   58.58  934.53   60.01
 1069.55   60.69 1187.17   58.03 1234.59   59.62 1327.77    59.7 1620.84   57.25
  1652.2   46.68 1653.28   42.68 1659.91   42.67  1660.9   46.57 1708.37   60.22
 1964.03   58.13 2010.35   55.86 2072.12   56.76 2303.74    56.8 2518.15   54.31
 2562.69   55.75 2848.58    57.1 3043.83   56.65 3277.43   58.22 3650.12   58.48
#Mann= 3 , 0 , 0
       0     .12       0 1620.84     .04       0 1708.37     .15       0
#XS Ineff= 2 , 0
       0    1593            1715       0
Permanent Ineff=
       T       T
Bank Sta=1620.84,1708.37
XS Rating Curve= 0
Exp/Cntr=.3,.1

Type RM Length L Ch R = 1 ,16158   ,47.77,52.07,58.99
BEGIN DESCRIPTION:
16157.68--u/s approach Chimney Rock West bridge; channel copied from 15814; blocked obstruction in D139 channel
END DESCRIPTION:
XS GIS Cut Line= 6
     3086283.788    13803570.887     3086319.846    13802191.669
     3085853.052    13801742.939     3085854.088     13801643.54
     3085657.754    13801358.719      3085917.02    13799887.126
#Sta/Elev= 30
       0   57.27  479.72   61.72  638.61   61.19  668.62   63.03  728.31    63.2
  933.03   60.58 1313.23   59.86 1436.21   56.06 1544.43   55.16 1739.23   56.79
 1819.89   59.77 1923.92   57.19 1998.96   58.71 2020.85    56.5 2074.85   42.41
 2080.76   42.47 2108.58    55.4 2127.86   58.03    2489   57.33 2565.15   54.76
  2745.3   54.98 2763.15   52.28 2778.38   55.29 2793.62   55.29 2824.08   51.23
 2861.85   54.63 2900.23   55.07 3067.77   54.15  3326.7   57.21 3966.78   59.53
#Mann= 3 , 0 , 0
       0      .1       0 1998.96     .04       0 2127.86      .1       0
#XS Ineff= 2 , 0
       0    1937            2161       0
Permanent Ineff=
       T       T
#Block Obstruct= 1 ,-1
 2745.12 2887.81   54.92
Bank Sta=1998.96,2127.86
XS Rating Curve= 0
Exp/Cntr=.5,.3

Type RM Length L Ch R = 1 ,16106   ,42.2,49.1,61.38
BEGIN DESCRIPTION:
16105.60--u/s face Chimney Rock West bridge; channel copied from 15814; blocked obstruction in D139 channel
END DESCRIPTION:
XS GIS Cut Line= 6
     3086335.365    13803588.931     3086371.847    13802193.979
     3085905.053    13801745.249     3085906.089     13801645.85
     3085709.755    13801361.029     3085965.328    13799910.482
#Sta/Elev= 30
       0   56.71   26.44   56.15   66.84   57.96  431.58   61.61  701.67   61.04
  746.69    62.8  929.58   60.44 1241.86   59.57 1368.26   55.59 1628.44    54.8
 1782.92   55.98 1844.88   57.81 1866.14   56.89 1949.37    57.7 1970.18   56.53
 2039.68   57.92  2093.9   42.79 2098.85   42.41 2104.76   42.47 2130.68   54.23
 2488.27   56.62 2562.75   53.98 2653.39   54.32 2705.08   48.85 2756.99   55.45
 2847.64   54.79 3009.71   56.34 3070.63   55.44 3310.92   55.42 3961.16   59.78
#Mann= 3 , 0 , 0
       0      .1       0 2039.68     .04       0 2130.68      .1       0
#XS Ineff= 2 , 0
       0    1960            2199       0
Permanent Ineff=
       T       T
#Block Obstruct= 1 ,-1
 2640.49 2754.99   54.67
Bank Sta=2039.68,2130.68
XS Rating Curve= 0
Exp/Cntr=.5,.3

Type RM Length L Ch R = 3 ,16082   ,,,
BEGIN DESCRIPTION:
Chimney Rock West (U/S) Bridge
END DESCRIPTION:
Bridge Culvert--1,0,-1,-1, 0
Deck Dist Width WeirC Skew NumUp NumDn MinLoCord MaxHiCord MaxSubmerge Is_Ogee
5,38,2.6,0, 7, 7, , , .95, 0, 0,0,,
    2040 2070.28 2070.28 2098.83 2127.37 2127.37 2164.62
   55.03   55.03   55.03   55.02   55.09   55.09   54.57
     -.1     -.1   53.44   53.57   53.44     -.1     -.1
    2056 2086.28 2086.28 2114.83 2143.37 2143.37 2180.62
   55.03   55.03   55.03   55.02   55.09   55.09   54.57
     -.1     -.1   53.44   53.57   53.44     -.1     -.1
Pier Skew, UpSta & Num, DnSta & Num=  ,2089.31, 2 ,2105.31, 2 , 0 , 0 , 0 ,,
     .63     .63
       0   53.57
     .63     .63
       0   53.57
Pier Skew, UpSta & Num, DnSta & Num=  ,2108.34, 2 ,2124.34, 2 , 0 , 0 , 0 ,,
     .63     .63
       0   53.57
     .63     .63
       0   53.57
BR Coef=-1 , 1 , 1 ,1.05, 0 ,,,.8,-1,1.2,0,
WSPro=,,,, 1 ,,,, 0 ,,,, 0 ,,,,-1 ,-1 ,-1 , 0 , 0 , 0 , 0 , 0
BC Design=,, 0 ,, 0 ,,,,,,

Type RM Length L Ch R = 1 ,16057   ,104.67,119.67,164.93
BEGIN DESCRIPTION:
16056.51--d/s face Chimney Rock West bridge; channel copied from 15814; blocked obstruction in D139 channel
END DESCRIPTION:
XS GIS Cut Line= 6
     3086383.655    13803605.824     3086420.718    13802189.299
     3085953.924    13801740.569      3085954.96     13801641.17
     3085758.626    13801356.349     3086009.621    13799931.897
#Sta/Elev= 30
       0    56.4  387.17   61.64  778.59   62.02  913.59   59.77 1213.74   59.53
  1308.4   56.36 1381.51   56.91 1476.96   55.05 1643.26   56.83 1686.55   55.48
 2064.51    55.6  2109.9   42.79 2114.85   42.41 2120.76   42.47 2147.58   54.77
 2150.27   54.86 2238.73   55.56    2564   54.54 2589.89    53.6 2628.74   48.62
 2645.76   50.51 2654.64   53.21 2693.49   55.46 2843.76   54.23 2877.93   56.04
 3081.97   56.14 3163.62   57.87  3405.7   58.05 3468.24    56.5 3956.24   59.78
#Mann= 3 , 0 , 0
       0      .1       0 2064.51     .04       0 2150.27      .1       0
#XS Ineff= 2 , 0
       0    1983            2229       0
Permanent Ineff=
       T       T
#Block Obstruct= 1 ,-1
 2551.04 2680.75   54.65
Bank Sta=2064.51,2150.27
XS Rating Curve= 0
Exp/Cntr=.5,.3

Type RM Length L Ch R = 1 ,15937   ,44.83,49.1,59.18
BEGIN DESCRIPTION:
15936.84--u/s face Chimney Rock East bridge; channel & LOB copied from 15814; blocked obstruction in D139 channel
END DESCRIPTION:
XS GIS Cut Line= 6
     3086501.367    13803647.005     3086539.841    13802177.889
     3086073.047    13801729.159     3086074.083     13801629.76
     3085877.749    13801344.939     3086117.584    13799984.095
#Sta/Elev= 30
       0   56.44   84.53    56.1   137.1   58.72   268.7   60.61  324.62   59.54
  489.67   61.55  819.79   62.12  969.84   59.68 1089.88    59.9 1189.89   58.41
 1248.38   56.35 1314.96   56.69 1336.12   54.41 1365.36   48.82 1379.98   48.65
 1409.23   54.79 1423.85   56.77 1438.47   57.15 1942.85   55.75 2112.85    56.5
  2161.9   42.79 2166.85   42.41 2172.76   42.47 2192.45   51.46 2203.78   54.11
 2879.44   55.05 3008.93   58.02 3387.42   58.49 3494.04   56.86 3944.27   59.26
#Mann= 3 , 0 , 0
       0      .1       0 2112.85     .04       0 2203.78      .1       0
#XS Ineff= 2 , 0
       0    2049            2305       0
Permanent Ineff=
       T       T
#Block Obstruct= 1 ,-1
 1292.13 1438.48   57.15
Bank Sta=2112.85,2203.78
XS Rating Curve= 0
Exp/Cntr=.5,.3

Type RM Length L Ch R = 3 ,15913   ,,,
BEGIN DESCRIPTION:
Chimney Rock East (D/S) Bridge
END DESCRIPTION:
Bridge Culvert--1,0,-1,-1, 0
Deck Dist Width WeirC Skew NumUp NumDn MinLoCord MaxHiCord MaxSubmerge Is_Ogee
5,38,2.6,0, 7, 7, , , .95, 0, 0,0,,
    2110 2138.61 2138.61 2166.83 2195.04 2195.04 2263.36
   54.96   54.96   54.96   55.09   55.05   55.05   54.36
     -.1     -.1   53.32   53.45   53.41     -.1     -.1
    2145 2173.61 2173.61 2201.83 2230.04 2230.04 2298.36
   54.96   54.96   54.96   55.09   55.05   55.05   54.36
     -.1     -.1   53.32   53.45   53.41     -.1     -.1
Pier Skew, UpSta & Num, DnSta & Num=  ,2157.42, 2 ,2192.42, 2 , 0 , 0 , 0 ,,
     .63     .63
       0   53.57
     .63     .63
       0   53.57
Pier Skew, UpSta & Num, DnSta & Num=  ,2176.23, 2 ,2211.23, 2 , 0 , 0 , 0 ,,
     .63     .63
       0   53.57
     .63     .63
       0   53.57
BR Coef=-1 , 1 , 1 ,1.05, 0 ,,,.8,-1,1.2,0,
WSPro=,,,, 1 ,,,, 0 ,,,, 0 ,,,,-1 ,-1 ,-1 , 0 , 0 , 0 , 0 , 0
BC Design=,, 0 ,, 0 ,,,,,,

Type RM Length L Ch R = 1 ,15888   ,111.59,73.35,83.18
BEGIN DESCRIPTION:
15887.75--d/s face Chimney Rock East bridge; channel copied from 15814; blocked obstruction in D139 channel
END DESCRIPTION:
XS GIS Cut Line= 6
     3086549.657    13803663.898     3086588.712    13802173.209
     3086121.918    13801724.479     3086122.954     13801625.08
      3085926.62    13801340.259     3086161.876    13800005.509
#Sta/Elev= 30
       0   56.34  116.44   56.91  176.46   59.25  221.47   59.56   296.5   58.55
  551.59    61.5   872.2   61.71 1106.78   59.23 1217.76   56.59 1276.25   57.05
 1290.88   56.22 1320.12   49.93 1334.74   48.24 1349.36   49.31 1378.61   57.13
 1406.88   57.76  1491.2   55.82 1521.08    56.7 1845.75   54.77 2137.89   55.68
 2147.85    56.5  2196.9   42.79 2201.85   42.41 2207.76   42.47 2235.58    55.4
 2855.92   54.96 3008.24   57.99  3526.1   57.02 3631.72   58.48 3939.36   58.93
#Mann= 3 , 0 , 0
       0      .1       0 2147.85     .04       0 2235.58      .1       0
#XS Ineff= 2 , 0
       0    2072            2338       0
Permanent Ineff=
       T       T
#Block Obstruct= 1 ,-1
  1271.7 1383.77   57.13
Bank Sta=2147.85,2235.58
XS Rating Curve= 0
Exp/Cntr=.5,.3

Type RM Length L Ch R = 1 ,15814   ,269.45,147.57,310.3
BEGIN DESCRIPTION:
15814.39--d/s exit Chimney Rock East bridge; surveyed channel; blocked obstruction in D139 channel
END DESCRIPTION:
XS GIS Cut Line= 6
     3086621.014    13803678.321     3086661.738    13802165.516
     3086194.944    13801716.786      3086195.98    13801617.387
     3085999.646    13801332.566     3086229.137    13800024.569
#Sta/Elev= 30
       0   55.87  100.86   58.07  265.92    57.3  641.05   61.71  836.12   61.74
  1046.2   59.08 1146.86   56.13 1205.31      57 1219.92   56.51 1263.76    48.3
 1271.28    48.3 1278.37   48.33 1322.21   58.01 1380.65   56.47    1662   56.77
 1699.56   55.54 2160.85    56.5  2209.9   42.79 2214.85   42.41 2220.76   42.47
 2248.58    55.4  2466.6    56.5 2870.23   54.79 2992.06   58.26 3098.67   59.35
 3209.01   59.43 3260.83   57.06 3768.75   59.62 3814.44   58.58 3934.17   58.72
#Mann= 3 , 0 , 0
       0      .1       0 2160.85     .04       0 2248.58      .1       0
#XS Ineff= 2 , 0
       0    2095            2366       0
Permanent Ineff=
       T       T
#Block Obstruct= 1 ,-1
  1190.6 1326.19   57.17
Bank Sta=2160.85,2248.58
XS Rating Curve= 0
Exp/Cntr=.3,.1

Type RM Length L Ch R = 1 ,15667   ,534.67,694.47,681.43
BEGIN DESCRIPTION:
15666.83--surveyed channel; blocked obstruction in D139 channel & anamolous hole in apt. parking lot
END DESCRIPTION:
XS GIS Cut Line= 5
     3086775.326    13803742.847     3086801.067     13802011.71
     3086340.827    13801706.049     3086344.064    13801603.578
     3086680.771    13800256.382
#Sta/Elev= 30
       0   55.84  155.23   58.53  390.39   57.16  923.89   61.24   997.8   59.57
 1056.92   55.38 1130.83   56.46 1175.18   48.23 1189.96   48.83 1219.52   56.39
 1249.09   57.53 1293.43   55.78 1633.42    57.4 1775.09   55.52 2283.82   56.22
 2340.61   43.23 2347.87   43.59 2373.28   55.21 2386.35   56.46 2392.61   52.93
 2408.07   50.93 2438.99   50.31 2485.38   51.58  2516.3   56.35 2531.76   56.79
 2810.07   56.21 2913.72   54.13 3505.83   60.21 3567.68    58.6 3774.98    60.6
#Mann= 3 , 0 , 0
       0      .1       0 2283.82     .04       0 2373.28      .1       0
#XS Ineff= 2 , 0
       0    2205            2437       0
Permanent Ineff=
       T       T
#Block Obstruct= 2 ,-1
  1130.8 1221.02    56.4 2386.35 2523.65   56.42
Bank Sta=2283.82,2373.28
XS Rating Curve= 0
Exp/Cntr=.3,.1
